--- sycmrcrk.prj (project) ---

Proj Title=sycmrcrk
Current Plan=p01
Default Exp/Contr=0,0
English Units
Geom File=g01
Flow File=f01
Plan File=p01
BEGIN DESCRIPTION:
END DESCRIPTION:
DSS Export Rating Curves= 0
DSS Export Rating Curve Sorted= 0
DSS Export Volume Flow Curves= 0
DXF OffsetX= 0
DXF OffsetY= 0
DXF ScaleX= 0
DXF ScaleY= 0

--- sycmrcrk.p01 (plan) ---

Plan Title=Floodplain
Program Version=4.00
Geom File=g01
Flow File=f01
K Sum by GR=0
Std Step Tol=0.01
Critical Tol=0.01
Num of Std Step Trials=20
Max Error Tol=0.3
Flow Tol Ratio=0.001
Split Flow NTrial=30
Split Flow Tol=0.02
Split Flow Ratio=0.02
Log Output Level=0
Friction Slope Method=1
Unsteady Friction Slope Method=2
Unsteady Bridges Friction Slope Method=1
Global Log Level=0
CheckData=False
Run HTab=0
Run UNet=0
Run PostProcess=0
UNET Theta=0
UNET Theta Warmup=0
UNET ZTol=0
UNET ZSATol=0
UNET MxIter=0
UNET MaxInSteps=0
UNET DtIC=0
UNET DtMin=0
UNET MaxCRTS=0
UNET WFStab=0
UNET SFStab=0
UNET WFX=0
UNET SFX=0
UNET DSS MLevel=0
UNET DZMax Abort=0
UNET Convert EG Bridges=0
UNET Use Existing IB Tables=0
UNET Froude Limit=0
UNET Froude Power=0
Write IC File=0
Echo Input=False
Echo Output=False
Write Detailed=0

--- sycmrcrk.f01 (steady flow) ---

Flow Title=NFF Regression Equation
Program Version=4.00
Number of Profiles= 1
Profile Names=P100yr
River Rch & RM=sycmrcrk,Main            ,10691.4
     355
River Rch & RM=sycmrcrk,Main            ,9594.6
     374
River Rch & RM=sycmrcrk,Main            ,8911.5
     412
River Rch & RM=sycmrcrk,Main            ,7685.2
     427
River Rch & RM=sycmrcrk,Main            ,7390.7
     517
River Rch & RM=sycmrcrk,Main            ,5633.9
     540
River Rch & RM=sycmrcrk,Main            ,5407
     661
River Rch & RM=sycmrcrk,Main            ,4802.6
     679
River Rch & RM=sycmrcrk,Main            ,3812.2
     742
River Rch & RM=sycmrcrk,Main            ,1192.2
     792
Boundary for River Rch & Prof#=sycmrcrk,Main            , 1
Up Type= 0
Dn Type= 3
Dn Slope=0.010018
DSS Import GetInterval= 0
DSS Import GetPeak= 0
DSS Import FillOption= 0

--- sycmrcrk.g01 (geometry) ---

Geom Title=USGS 10m DEM
Program Version=4.00

River Reach=sycmrcrk        ,Main
Reach XY= 30
     1611829.095      252587.185     1611302.342      252322.353
     1611040.015      252000.221     1611026.189      251807.947
     1610830.658      251534.782     1610718.838      251278.868
     1610684.385      250720.532     1610634.241      250653.134
     1610686.513      250509.097     1610646.766      250253.718
     1610442.328      250221.824     1610369.956      250092.952
     1610042.251      249787.393      1610044.91      249597.867
     1609980.416      249498.978     1609747.485      249423.769
     1609160.719      248926.642      1609136.65      247964.069
     1608841.829      247424.209     1608661.292       246936.84
     1608534.119      246753.704     1608318.178      246561.801
     1608294.212      246424.828     1608220.132      246393.773
     1608195.291      246115.853     1608100.482      246001.137
     1607679.036      245532.372     1607115.223      245183.638
     1606857.509      244620.648     1606791.562      244226.575

Type RM Length L Ch R = 1 ,10691.4 ,90.3,105.5,120.6
XS GIS Cut Line= 4
     1611944.015      252276.397     1611812.464      252527.792
     1611827.827      252656.071     1611825.437      252848.233
#Sta/Elev= 30
    10.1 1046.97    20.3 1040.82    70.9 1006.23    91.2  988.45   101.3   983.7
   121.6  966.04   162.1  928.88   182.4  911.74   192.5  904.28   202.7  901.89
   222.9  887.12   233.1  880.65   243.2  875.56   253.3  871.69   263.5  869.53
   283.7  867.55   323.5  867.16   333.4  866.26   343.4  865.42   353.4  865.77
   373.2  868.55   412.9  877.13   443.3  879.09   483.7   879.8   493.8  881.79
     504  886.55   514.1  892.54   524.2  893.91   534.3  898.44   605.1  936.18
#Mann= 3 , 0 , 0
       0     .06       0   333.4    .045       0   353.4     .06       0
Bank Sta=333.4,353.4
XS Rating Curve= 0 ,0
Exp/Cntr=0.3,0.1

Type RM Length L Ch R = 1 ,10586   ,143.5,143.2,142.8
XS GIS Cut Line= 4
     1611888.254      252273.325     1611781.739      252480.892
     1611691.611      252602.429     1611574.171      252788.148
#Sta/Elev= 30
     9.7 1012.87    38.9 1000.39    48.6  994.66    77.8  972.56    87.5  969.71
    97.2  963.77   106.9  955.83   136.1  926.65   155.5   910.2     175  895.25
   194.4  882.72   204.1  881.14   223.6  871.41   233.3   869.5  320.01   862.3
   334.2  861.68  340.39  862.74   344.3  863.76   364.4  874.91   404.6  875.92
   414.6   878.7   424.6  883.98   444.5  889.84   484.5  907.39   514.5  923.02
   534.4  935.07   544.4  937.28   564.4  952.33   584.4  964.16   604.3  978.64
#Mann= 3 , 0 , 0
     9.7     .06       0  320.01    .045       0  340.39     .06       0
Bank Sta=320.01,340.39
XS Rating Curve= 0 ,0
Exp/Cntr=0.3,0.1

Type RM Length L Ch R = 1 ,10442.8 ,182.5,180.2,178
XS GIS Cut Line= 4
     1611766.718      252244.647     1611645.181      252424.904
     1611576.902       252521.86     1611485.408      252669.342
#Sta/Elev= 30
     9.9  948.59    19.8  943.51    39.5  930.39    49.4  925.74    88.9  908.28
   108.7  900.51   118.6  897.72   128.5  892.96   138.3  887.27   158.1  871.16
     168  868.62   217.4  863.85     247  861.92  262.88  859.63   276.7  858.35
  283.65  859.53   286.7  860.08   306.3  869.06   316.2  872.16   326.1  872.93
   355.3     873   364.9  873.88   384.2   888.4   393.8   894.8   403.5  899.99
   413.1     903   432.4  906.35   461.3  914.07   480.6  922.47   509.5  939.68
#Mann= 3 , 0 , 0
     9.9     .06       0  262.88    .045       0  283.65     .06       0
Bank Sta=262.88,283.65
XS Rating Curve= 0 ,0
Exp/Cntr=0.3,0.1

Type RM Length L Ch R = 1 ,10262.6 ,185,190.2,195.3
XS GIS Cut Line= 4
     1611585.096      252149.057     1611492.236      252315.658
     1611425.323      252437.194     1611362.506      252557.365
#Sta/Elev= 30
      10  944.69    40.2  928.39    50.2   922.4    60.2  913.26    70.3  902.94
    80.3  898.28    90.3  888.84   100.4  881.92   120.5  870.48   130.5  865.67
   140.5  863.55   150.6  862.45   170.7  860.73   190.7  859.62  264.55  853.55
   279.9  853.08  282.88  853.96   289.8  856.49   299.7  857.86   319.6  867.87
   329.5  869.31   339.2  869.41   348.8  871.31   358.5  877.57   397.3  906.38
     407  908.02   426.3  922.22     436  928.65   445.7  934.57   465.1  945.19
#Mann= 3 , 0 , 0
      10     .06       0  264.55    .045       0  282.88     .06       0
Bank Sta=264.55,282.88
XS Rating Curve= 0 ,0
Exp/Cntr=0.3,0.1

Type RM Length L Ch R = 1 ,10072.4 ,252.2,255.4,258.6
XS GIS Cut Line= 4
     1611490.871      252064.391     1611367.969       252215.97
     1611257.357      252332.045     1611124.896      252457.678
#Sta/Elev= 30
     9.8  923.04    29.3  915.37      39  912.92    48.8  911.11    87.8  895.79
    97.6  890.33   146.4  865.09   156.1  860.56   165.9  857.77   185.4   856.4
   205.2  854.39  300.22   848.4   315.4  847.79  320.09  848.58   325.4  849.65
   345.5  858.81   355.5  862.84   365.1  865.06   374.7  866.29   384.3   870.9
   393.9  879.05   413.1  891.62   422.7  895.54   432.4  898.35   461.2  916.78
   470.8  922.95   480.4  930.08     490  938.99   509.2  951.66     538  969.66
#Mann= 3 , 0 , 0
     9.8     .06       0  300.22    .045       0  320.09     .06       0
Bank Sta=300.22,320.09
XS Rating Curve= 0 ,0
Exp/Cntr=0.3,0.1

Type RM Length L Ch R = 1 ,9817    ,212.5,222.4,232.3
XS GIS Cut Line= 4
     1611355.678       251919.64     1611200.002       252049.37
     1611074.369       252144.96     1610966.489      252258.303
#Sta/Elev= 30
    10.1  976.01    20.3  968.34    30.4  957.61    70.9  930.37    81.1  924.87
    91.2  921.18   101.3  914.93   111.5  908.07   121.6  897.78   131.7  890.22
   192.5   854.9   202.6   850.2   212.5  847.34   222.4  846.11   301.2  843.44
   311.2  843.14   321.2  843.88   330.9  847.48   340.8  853.65   350.6  857.48
   370.3  860.38   380.1  864.07   399.6     873     429  887.59   468.1  903.56
   477.9  909.32   487.6  916.19   497.4  920.55   507.2  922.26     517  926.76
#Mann= 3 , 0 , 0
       0     .06       0   301.2    .045       0   321.2     .06       0
Bank Sta=301.2,321.2
XS Rating Curve= 0 ,0
Exp/Cntr=0.3,0.1

Type RM Length L Ch R = 1 ,9594.6  ,203.5,196,188.4
XS GIS Cut Line= 4
     1611295.593      251815.856     1611063.445      251910.081
     1610971.951      251925.102      1610817.64      252060.294
#Sta/Elev= 30
      10  984.89    50.1  959.97    60.1  949.38    80.2  936.07   110.2  915.19
   120.3  909.73   130.3  902.22   140.3  892.87   160.3  881.22   200.4  859.62
   210.5  850.87   220.5  846.35   230.5  844.83   269.1   841.4   278.4  840.24
   286.9  838.42   296.9  837.87   306.9  838.86     334  845.79   362.8  849.67
   382.3  851.51   392.1  853.35     441  874.39   460.5  886.84     480  896.29
   489.8  900.32   499.6  902.85   509.3  907.21   538.6  921.61   548.4  928.69
#Mann= 3 , 0 , 0
       0     .06       0   286.9    .045       0   306.9     .06       0
Bank Sta=286.9,306.9
XS Rating Curve= 0 ,0
Exp/Cntr=0.3,0.1

Type RM Length L Ch R = 1 ,9398.6  ,168.9,169.9,170.9
XS GIS Cut Line= 4
     1611167.229      251639.696     1611042.961      251698.416
     1610915.962      251774.888     1610787.598      251971.532
#Sta/Elev= 30
     9.8   943.5    19.6  936.39    29.5  932.68    39.3  928.42    88.4  901.82
    98.2  893.26     108  887.31   147.3  861.91   167.1  850.14     177  841.64
   186.9  836.28   196.7  833.98   206.5  832.88   216.5  832.73   226.5  833.55
   246.2  835.98   265.9  836.48   275.8  837.17   334.6   844.7   354.2  845.96
     364  847.37   373.8   851.1   383.5  857.29   393.3   861.4   442.2  876.38
     452  878.08   461.8  880.45   471.6  885.18   491.2  897.53   520.5  910.81
#Mann= 3 , 0 , 0
       0      .1       0   206.5    .045       0   226.5      .1       0
Bank Sta=206.5,226.5
XS Rating Curve= 0 ,0
Exp/Cntr=0.3,0.1

Type RM Length L Ch R = 1 ,9228.7  ,167.6,169,170.4
XS GIS Cut Line= 4
      1611086.66      251516.794     1610940.543       251567.32
      1610780.77      251653.352     1610629.191      251725.728
#Sta/Elev= 30
     9.7  961.25    19.3  955.84      29  946.43    48.3  938.58      87  915.22
    96.6  908.45   106.3  898.06   154.6  872.93   164.7  867.14   174.8  859.61
   184.8  850.09   194.9  843.32     205  835.57   215.1  829.29  221.33  828.12
   225.2  827.41  242.38   827.6     326   830.5   336.1  831.46   355.8  837.63
   365.7  839.94   385.5   841.3   405.2  840.67   415.1  843.38     425  848.66
   434.9  850.81   444.8  855.92   484.3  878.32   494.2  885.56     504   893.8
#Mann= 3 , 0 , 0
     9.7      .1       0  221.33    .045       0  242.38     .08       0
Bank Sta=221.33,242.38
XS Rating Curve= 0 ,0
Exp/Cntr=0.3,0.1

Type RM Length L Ch R = 1 ,9059.7  ,144.8,148.2,151.6
XS GIS Cut Line= 4
     1610997.897      251377.505     1610861.339        251425.3
     1610712.491      251492.214     1610570.471      251546.837
#Sta/Elev= 30
     9.6  954.34    19.3  948.07    28.9   938.1    38.6  929.22    67.5  910.31
    77.2  903.18    86.8  895.54    96.5  891.46   106.1  883.99   115.7  878.35
     135     869   173.5  849.61   183.1  840.93   202.3  828.69   211.9  823.41
  217.34  822.07   221.5  821.14  237.94  821.88   259.9  823.79   288.7  825.53
   317.4  826.56   326.9  826.15   345.9  831.96   355.4  833.12   364.9  833.22
   374.4  834.01     384  836.74     403  844.76     422  856.44     460  872.15
#Mann= 3 , 0 , 0
     9.6      .1       0  217.34    .045       0  237.94      .1       0
Bank Sta=217.34,237.94
XS Rating Curve= 0 ,0
Exp/Cntr=0.3,0.1

Type RM Length L Ch R = 1 ,8911.5  ,237,240.8,244.6
XS GIS Cut Line= 4
     1610974.682      251269.624     1610806.716      251302.398
     1610634.653      251347.462     1610476.246      251410.279
#Sta/Elev= 30
    10.1  952.65    20.1     941    50.3  921.74    90.6  896.75   130.9  876.78
   140.9   872.9   161.1     864   171.1  855.82     181  849.94   210.7  835.89
   220.5  830.95   240.3  819.63  246.79  817.39   250.2  816.16   269.9  817.09
   309.5  820.49   319.4  821.81   329.2  821.87   339.1  822.54     349  824.58
     369  829.52   379.1  833.26   399.1  845.66   409.1  848.62   419.2  851.11
   439.2  856.67   459.3  861.19   469.3   864.9   499.4  872.31   519.4  879.26
#Mann= 3 , 0 , 0
    10.1      .1       0  246.79    .045       0   269.9     .06       0
Bank Sta=246.79,269.9
XS Rating Curve= 0 ,0
Exp/Cntr=0.3,0.1

Type RM Length L Ch R = 1 ,8670.7  ,208.2,207.7,207.2
XS GIS Cut Line= 4
     1610932.349      251071.616     1610798.522      251079.809
     1610586.858       251094.83     1610446.203      251164.475
#Sta/Elev= 30
     9.6  951.66    38.3  935.42    57.5  921.56      67  916.51    76.6  908.64
    86.2  902.42   105.3  889.14   134.1  872.51   154.3  854.95   194.7  831.27
   204.8  824.59   214.9  816.62  222.31  813.24     225   812.1  241.96   812.6
   285.6  814.22   305.9  815.83   336.2  817.29   346.3  818.38   365.9  822.15
   375.7  823.51   385.5  826.28   395.3  829.85   434.6  845.04   444.4  849.32
   454.2  856.66     464  861.52   483.6  869.15   493.4  873.48   503.2  878.49
#Mann= 3 , 0 , 0
     9.6      .1       0  222.31    .045       0  241.96     .06       0
Bank Sta=222.31,241.96
XS Rating Curve= 0 ,0
Exp/Cntr=0.3,0.1

Type RM Length L Ch R = 1 ,8463    ,191.9,190.9,190.6
XS GIS Cut Line= 4
     1610872.264       250869.51     1610776.673      250877.703
     1610528.138      250898.187     1610412.064      250959.638
#Sta/Elev= 30
     9.6  921.76    19.2  915.87    28.8   909.6    38.4  899.41    57.6  890.99
    67.2   886.2    95.9  871.39   105.9  862.64   115.9  855.91   145.8  840.82
   165.8  830.48   175.7  825.14   185.7  815.53   195.7  808.23   205.7  807.07
   215.7  807.42   235.6  808.25   295.4  809.34   305.4  809.84   315.4   811.2
   335.3  816.14   345.3   816.5   355.4  817.79   365.5  820.72   395.8  830.86
   405.9  834.54     416  840.24   426.1  844.23   446.3  850.43   476.7  860.64
#Mann= 3 , 0 , 0
       0      .1       0   195.7    .045       0   215.7      .1       0
Bank Sta=195.7,215.7
XS Rating Curve= 0 ,0
Exp/Cntr=0.3,0.1

Type RM Length L Ch R = 1 ,8272    ,239.6,241.5,241.9
XS GIS Cut Line= 4
     1610869.532      250676.963     1610747.996      250690.619
     1610522.676      250719.296     1610386.118      250801.231
#Sta/Elev= 30
     9.4  928.25    18.8  921.76    37.6  909.13      47   902.1    56.4   891.9
    65.9  886.35    84.7   873.7   112.9  854.34   122.3  844.74   132.2  834.99
   142.1  829.03   151.9  823.47   181.6   807.2   191.3  803.71   201.3  802.64
   211.3  803.22   319.8  805.47   329.7  805.78   339.6  806.69   349.4  809.19
   359.4  810.85   369.3  811.15   379.3  811.77   389.3  813.59   399.2  817.06
   419.1  824.99     439  836.76   468.9  848.37   498.7  860.46   508.7  865.84
#Mann= 3 , 0 , 0
       0      .1       0   191.3    .045       0   211.3     .08       0
Bank Sta=191.3,211.3
XS Rating Curve= 0 ,0
Exp/Cntr=0.3,0.1

Type RM Length L Ch R = 1 ,8030.5  ,114.6,112.7,110.8
XS GIS Cut Line= 4
     1610881.823      250478.954     1610758.921      250478.954
     1610596.417      250496.707     1610380.656      250592.298
#Sta/Elev= 30
     9.5  936.96    18.9  926.61    47.3  908.73    56.7  902.63    75.6  891.04
    85.1  880.05    94.5  872.02   151.7  832.93   161.4  824.91     171  813.23
   180.6  805.76   190.2  799.51  196.32  797.68   199.8  796.75   219.1  797.13
   228.7  797.46   238.3  798.14   296.2  801.25     306   802.1   315.9  803.33
     365  807.07   374.9  807.63   384.7   807.4   394.5  806.22   414.2  806.14
     424  807.16   433.9  810.73   463.4  825.07     483  839.63   522.4  858.42
#Mann= 3 , 0 , 0
     9.5      .1       0  196.32    .045       0   219.1     .06       0
Bank Sta=196.32,219.1
XS Rating Curve= 0 ,0
Exp/Cntr=0.3,0.1

Type RM Length L Ch R = 1 ,7917.8  ,255,232.6,210.3
XS GIS Cut Line= 4
     1610892.747      250391.557     1610728.878      250364.246
     1610547.256      250401.116     1610398.408      250518.556
#Sta/Elev= 30
     9.8  928.31    19.5  924.74    29.3  920.16    39.1  911.36      88  883.86
   107.5  872.13   117.3  861.49     127  852.98   146.6  840.55   166.1  830.44
   175.9  826.28   185.6  821.36   195.4  815.15   224.7  804.16   234.4  799.45
   244.2  795.41  247.72  794.86   253.9  793.94   273.4  794.43   331.9  796.72
   391.4  800.74   421.3  801.44   441.3  803.42   461.2  804.79   471.2  807.74
   481.2  811.95   501.1  821.21   511.1   829.7   521.1  835.93   541.1  845.42
#Mann= 3 , 0 , 0
     9.8      .1       0  247.72    .045       0   273.4     .06       0
Bank Sta=247.72,273.4
XS Rating Curve= 0 ,0
Exp/Cntr=0.3,0.1

Type RM Length L Ch R = 1 ,7685.2  ,286.3,294.5,302.4
XS GIS Cut Line= 4
      1610722.05      249894.487     1610575.933       250137.56
     1610519.944      250335.569     1610369.731      250507.632
#Sta/Elev= 30
    10.1  892.12    40.5  872.48    50.6  869.83    60.8  865.82      81  853.77
   111.4  836.72   121.5  832.11   162.1  816.89   172.2  816.19   182.3  812.57
   212.7  799.44   222.8   797.9   253.2  795.49   361.8   789.3   371.8  789.27
   381.8  789.29   469.8  794.29   499.3  795.24     539  797.45     549  798.39
   568.8  801.83   588.7   803.4   598.6  804.95   608.6  807.37   618.5  810.49
   638.3  818.14   648.3  824.39   658.2  832.28   697.9  850.56   717.8  859.19
#Mann= 3 , 0 , 0
       0     .06       0   361.8    .045       0   381.8     .06       0
Bank Sta=361.8,381.8
XS Rating Curve= 0 ,0
Exp/Cntr=0.3,0.1

Type RM Length L Ch R = 1 ,7390.7  ,221.3,223,224.6
XS GIS Cut Line= 4
     1610582.761      249805.724     1610412.064      249983.249
     1610306.914      250115.711      1610249.56      250226.323
#Sta/Elev= 30
     9.9   880.8    19.7  874.49    29.6  868.88    39.4  864.42    78.8  842.23
    88.7  837.48   108.4  829.54   118.2  824.48   147.8  814.03   157.6  812.65
   167.5  809.87   206.9  796.39   216.7  792.36   226.6   790.8   286.1  788.22
     306  786.93   335.8  787.14  351.63  782.74   355.7  781.61   365.7  781.39
  369.95  782.53   375.6  784.06   385.6  788.16   415.4  792.97     425  798.57
   434.6  805.69   444.2  811.42   501.7  842.79   520.8  849.05     540  859.38
#Mann= 3 , 0 , 0
     9.9     .06       0  351.63    .045       0  369.95     .06       0
Bank Sta=351.63,369.95
XS Rating Curve= 0 ,0
Exp/Cntr=0.3,0.1

Type RM Length L Ch R = 1 ,7167.7  ,219.7,212,211.3
XS GIS Cut Line= 4
       1610450.3      249667.801     1610268.678      249828.939
     1610149.873      249955.938       1610073.4      250035.141
#Sta/Elev= 30
    10.1  875.64    40.5  859.69    60.7  852.21    70.8  845.15    91.1   834.5
   101.2  830.45   131.5  821.28   141.6  817.73   151.8  811.59   182.1  798.66
   202.3  792.42   212.5  788.43   222.6  785.89   232.7  784.88   310.4  781.29
   339.4  780.79   348.7  779.28   358.7  777.74   368.7  778.25   378.1  780.51
   387.7  783.38   397.4  785.52     407  786.77   416.7  790.22   426.7  795.63
   436.7  803.72   456.7  810.96   506.8  839.04   516.8  844.25   526.8  847.88
#Mann= 3 , 0 , 0
       0     .06       0   348.7    .045       0   368.7     .06       0
Bank Sta=348.7,368.7
XS Rating Curve= 0 ,0
Exp/Cntr=0.3,0.1

Type RM Length L Ch R = 1 ,6955.7  ,259.5,272.5,278.5
XS GIS Cut Line= 4
     1610302.818      249531.243     1610138.948      249659.607
     1609987.369      249823.477     1609920.456      249955.938
#Sta/Elev= 30
     9.9  884.76    59.5  854.77    69.4  851.97    79.3  845.39    89.2  837.59
     109  826.08   158.6  798.81   168.5  791.36   178.4  784.76   188.3  781.11
   198.2   780.5   208.2  780.53     247  781.63   256.7  781.32   314.9  777.65
   353.4  774.21   363.4   773.7   373.4  774.94   392.6  780.04   402.3  781.09
     412  783.43   461.1  807.88     471  810.28   480.9  816.12   500.6  826.27
   510.5  830.94   520.4  834.14   530.3  835.51   550.1  836.94   579.8  837.06
#Mann= 3 , 0 , 0
       0     .06       0   353.4    .045       0   373.4     .06       0
Bank Sta=353.4,373.4
XS Rating Curve= 0 ,0
Exp/Cntr=0.3,0.1

Type RM Length L Ch R = 1 ,6683.3  ,211.9,194.8,177.7
XS GIS Cut Line= 4
     1610266.896      249372.447     1610074.349      249465.306
     1609936.426      249554.069     1609738.417      249752.078
#Sta/Elev= 30
     9.7  945.37    38.9   924.6    58.3  905.21   116.6   876.9   126.3  871.06
     136  862.51   145.8  856.85   165.2  850.88   194.3  838.13   204.1  833.19
   213.8  825.91   252.4  807.72   271.7  796.27   281.3  789.15     291   778.7
  298.65  772.85   300.6  771.45   310.2  771.26  315.01  772.41   329.5  777.34
   339.2  778.99   467.8  773.26   527.8  776.94   547.8  784.56   567.8  794.83
   607.8  811.66   627.8  816.15   637.8  820.22   647.8  822.58   657.8  823.34
#Mann= 3 , 0 , 0
     9.7     .06       0  298.65    .045       0  315.01     .06       0
#XS Ineff= 2 , 0
       0                     339       0
Permanent Ineff=
       F       F
Bank Sta=298.65,315.01
XS Rating Curve= 0 ,0
Exp/Cntr=0.3,0.1

Type RM Length L Ch R = 1 ,6488.4  ,297.2,306.7,316.1
XS GIS Cut Line= 4
      1609943.68      249162.169     1609824.875      249396.707
     1609809.512      249501.174     1609723.481      249728.543
#Sta/Elev= 30
    10.1  937.47    60.7  901.93    70.8  896.76    80.9  893.68      91  884.06
   161.8  835.87   171.9  829.91     182  828.33   212.4  808.76   232.6  790.84
   252.8  778.03   262.9  773.61   272.5  771.82   291.7  773.16   301.3  771.06
   310.5  767.32   320.5  765.33   330.5  766.55   349.3  773.79   358.9  774.59
   429.3  771.61   459.7   774.4   479.9  774.92   490.1  778.41   500.2  780.04
   510.3  783.18   581.2  813.85   591.3  819.52   601.5  821.48   611.6  821.77
#Mann= 3 , 0 , 0
       0     .06       0   310.5    .045       0   330.5     .06       0
Bank Sta=310.5,330.5
XS Rating Curve= 0 ,0
Exp/Cntr=0.3,0.1

Type RM Length L Ch R = 1 ,6181.8  ,276.1,280.9,285.7
XS GIS Cut Line= 4
     1609747.027      249079.237     1609620.028      249228.085
       1609529.9      249353.718     1609461.621      249609.081
#Sta/Elev= 30
     9.8  902.56    19.6  894.02    58.7  870.21   107.6  843.42   127.2  829.35
   146.7   818.1   156.5  815.65   166.3  811.59   185.9   799.9     215  781.29
   234.3  765.52     244  761.66     263  759.02     273  758.76     283  759.01
   292.3  761.12   311.6  768.47   321.3  768.96   399.2  765.73     409  765.79
   418.8   767.4   477.6  793.51   487.3  794.32   516.7  807.47   526.5  810.67
   546.1  812.97   565.7  812.85   585.2   817.9     595  821.62   614.6  840.44
#Mann= 3 , 0 , 0
       0     .06       0     263    .045       0     283     .06       0
Bank Sta=263,283
XS Rating Curve= 0 ,0
Exp/Cntr=0.3,0.1

Type RM Length L Ch R = 1 ,5900.9  ,264.6,267,269.4
XS GIS Cut Line= 4
     1609577.695       248911.27     1609424.751      249060.119
     1609315.504      249154.343     1609221.279      249344.159
#Sta/Elev= 30
     9.7  914.41    29.1  895.14    38.8  887.49    58.2  874.93    77.6  864.01
    87.3  860.29      97  857.99   116.4  844.99     194  805.42   213.4  792.37
   232.7  786.29   251.9  774.18   271.1  758.07  275.49  756.32   280.7  754.15
   290.4  753.96  294.82  755.33   309.6   760.3   319.2  762.17     388  761.63
   428.3  762.64   438.4  765.66   458.6  774.23   468.7  776.06     499  791.01
   509.1  794.87   519.1  796.84   549.4  796.57   559.5  801.86   569.6   809.9
#Mann= 3 , 0 , 0
     9.7      .1       0  275.49    .045       0  294.82      .1       0
Bank Sta=275.49,294.82
XS Rating Curve= 0 ,0
Exp/Cntr=0.3,0.1

Type RM Length L Ch R = 1 ,5633.9  ,216.2,226.9,237.5
XS GIS Cut Line= 4
     1609468.449      248811.583     1609260.881      248873.034
      1609094.28      248985.012     1609042.389      249140.688
#Sta/Elev= 30
     9.8  899.63    49.2  878.57      59  872.69    78.7  856.37   118.1  834.52
   127.9  831.72   137.8  826.58   147.6  818.03   157.4  812.44   206.6  790.68
   216.5  785.55   226.5   777.9   256.6  760.04   266.7  756.24   296.8  753.43
   306.8  750.18   316.9  748.16   326.9  747.74   336.9  747.97     367  752.81
   377.1  755.37   397.1  762.25   407.2  763.66   465.5  764.79   475.1  766.27
   513.7  777.15   523.4  778.61     562  778.18   571.7  780.61   581.3  785.82
#Mann= 3 , 0 , 0
       0     .08       0   316.9    .045       0   336.9     .08       0
Bank Sta=316.9,336.9
XS Rating Curve= 0 ,0
Exp/Cntr=0.3,0.1

Type RM Length L Ch R = 1 ,5407    ,293.6,300,306.4
XS GIS Cut Line= 4
     1609497.126      248721.455     1609244.494      248706.434
      1609010.98      248722.821     1608721.478      248587.628
#Sta/Elev= 30
    10.1  924.78    20.2  918.41    30.4  905.89    40.5   899.5   101.2  866.35
   111.4  856.02   172.1  824.97   182.2  815.63   192.3  810.41   253.1  782.63
   262.8  774.36   272.6  769.21   301.8  756.03   330.9  745.02   340.9  743.26
   350.9   743.8   477.4  755.86   497.2  756.17   537.1  750.71   547.1  751.25
   557.1  754.22     567   759.7     577   769.1     617  789.96   656.9  812.93
   666.9  823.35   726.8  855.23   736.8  861.25   746.8   869.3   806.7  899.99
#Mann= 3 , 0 , 0
       0     .08       0   330.9    .045       0   350.9     .08       0
Bank Sta=330.9,350.9
XS Rating Curve= 0 ,0
Exp/Cntr=0.3,0.1

Type RM Length L Ch R = 1 ,5106.9  ,308.1,304.3,300.5
XS GIS Cut Line= 4
     1609465.718      248470.189     1609251.322      248434.684
     1609034.195      248381.426      1608810.24      248310.416
#Sta/Elev= 30
     9.9  867.58    19.8   862.5    29.6  852.84    98.8  817.09   118.5  802.01
   167.9  776.67   187.7  761.71   207.4  752.34   217.3  749.15     227  747.56
   275.6   746.3   295.1  740.12   304.5  738.24   314.5  737.81   324.5  738.35
     334  739.72   343.7  743.45   353.4  749.04   411.7  768.63   421.4  774.62
   431.2  778.83   499.6  804.22   509.4  810.82   577.9  835.52   587.7  840.73
   607.3  855.03   636.7  878.67   656.2  892.21     666  902.37   675.8  908.71
#Mann= 3 , 0 , 0
       0     .06       0   304.5    .045       0   324.5     .06       0
Bank Sta=304.5,324.5
XS Rating Curve= 0 ,0
Exp/Cntr=0.3,0.1

Type RM Length L Ch R = 1 ,4802.6  ,376.7,366.6,356.5
XS GIS Cut Line= 4
     1609603.641      248251.696     1609355.106      248134.256
     1609051.947      248116.504     1608833.455      248138.353
#Sta/Elev= 30
     9.8   828.3    39.3   820.9    98.2  802.89   127.6  792.04   147.3  782.12
   176.7  772.02   186.5  769.96   274.9  756.46   295.1  753.08   305.3  750.02
   335.6   745.6   355.9  744.31   457.1  744.14   467.2  742.91   477.5  739.45
   487.5  737.19   497.5  738.58   507.7  744.85     528  761.06   538.1  774.23
   568.4  795.66   598.5  815.01   608.5  823.57   658.4  840.94   678.4  851.25
   688.4   861.4   698.3  869.48   748.2  898.03   768.2  914.18   798.1  931.38
#Mann= 3 , 0 , 0
       0     .06       0   477.5    .045       0   497.5     .06       0
Bank Sta=477.5,497.5
XS Rating Curve= 0 ,0
Exp/Cntr=0.3,0.1

Type RM Length L Ch R = 1 ,4436.1  ,315.4,317.4,319.4
XS GIS Cut Line= 4
     1609494.395       247623.53     1609218.217      247695.538
     1608928.373      247833.803     1608782.929      247892.549
#Sta/Elev= 30
     9.8  862.56    29.5  853.22    68.9  839.08    88.6  827.32   137.8  807.43
   147.6   802.2   157.5  792.48   196.8  761.65   206.7  754.68   226.4  746.23
   255.9  740.44   295.4  737.23   345.6  736.91   415.9  738.85     446  736.87
     456   734.8     466  735.63   486.1  744.99   536.3  775.55   546.3  784.98
   556.4  792.35   586.5  810.26   596.5  815.71   616.3  822.93   626.2  830.86
   655.6  850.49   694.8  873.18   704.6  882.87   724.2  893.15   763.4  910.75
#Mann= 3 , 0 , 0
     9.8     .06       0     446    .045       0     466     .06       0
#XS Ineff= 2 , 0
       0     415                       0
Permanent Ineff=
       F       F
Bank Sta=446,466
XS Rating Curve= 0 ,0
Exp/Cntr=0.3,0.1

Type RM Length L Ch R = 1 ,4118.7  ,26.4,26.3,26.3
XS GIS Cut Line= 4
     1609480.739      247596.218     1609132.185      247415.936
      1608837.22      247522.451     1608711.918      247738.239
#Sta/Elev= 30
    10.1  848.68    90.6  822.27   130.8  817.96   140.9   814.7     161  803.41
   181.1  785.58   201.2  774.05   211.3  766.25   231.4  756.89   241.5  753.86
   271.7  750.15   382.4  742.03   422.8  736.14   453.1  733.48   544.2  732.96
   635.3  729.36   645.3  727.58   655.3  727.68     706  740.78     726  750.25
     736  751.11   765.9  765.86   785.9  773.89   805.8   787.2   815.8   791.8
   835.8   799.2   845.8  799.05   895.7  825.98   915.6  830.92   955.6     833
#Mann= 3 , 0 , 0
    10.1     .06       0   635.3    .045       0   655.3     .06       0
#XS Ineff= 2 , 0
       0     605             665       0
Permanent Ineff=
       F       F
Bank Sta=635.3,655.3
XS Rating Curve= 0 ,0
Exp/Cntr=0.3,0.1

Type RM Length L Ch R = 1 ,4092.3  ,28.8,28.8,28.9
XS GIS Cut Line= 4
     1609482.105      247583.928     1609118.871       247392.38
     1608792.488      247511.552     1608692.801      247735.507
#Sta/Elev= 30
      10  844.61    40.1  834.85    90.1   821.1   120.2  817.44   130.2  813.96
   170.3  793.34   220.3  760.42   230.4   755.9   240.4  753.86   410.6  741.49
   440.4  735.75   480.1  732.49     639  733.87   658.8  730.67   668.8  727.57
   678.8  730.32   688.6  734.26   718.4  735.13   748.2  740.14   777.7  743.37
   787.5  743.02   797.3  745.71   836.5  770.25   885.6  793.18   895.4   794.4
   905.2  797.75   934.6  816.23   954.2  826.76     964  829.59  1003.2  833.33
#Mann= 3 , 0 , 0
      10     .06       0   658.8    .045       0   678.8     .06       0
#XS Ineff= 2 , 0
       0     629                       0
Permanent Ineff=
       F       F
Bank Sta=658.8,678.8
XS Rating Curve= 0 ,0
Exp/Cntr=0.3,0.1

Type RM Length L Ch R = 1 ,4063.5  ,24.7,25.5,26.4
XS GIS Cut Line= 4
     1609482.105      247568.907     1609100.436      247369.847
     1608784.294      247484.241     1608529.965      247470.217
#Sta/Elev= 30
      10  839.45      40  830.56   110.1  814.84   130.1  805.86   150.2  801.28
   160.2  795.94   180.2  779.74   210.2  761.13   220.2  756.44   230.2  754.36
   410.4  743.08   440.3  739.55   460.1  735.18   509.6  731.35     648  735.19
   667.8  733.33  671.39  730.94   677.7  727.26   687.6   726.3  703.22  730.69
   796.1  742.66   815.6  748.29   825.4  752.48   835.2  760.27     894  783.98
   903.8   790.8   913.6  795.33   972.4  818.16     992  829.53  1021.4  840.44
#Mann= 3 , 0 , 0
      10     .06       0  671.39    .045       0  703.22     .06       0
#XS Ineff= 2 , 0
       0     648                       0
Permanent Ineff=
       F       F
Bank Sta=671.39,703.22
XS Rating Curve= 0 ,0
Exp/Cntr=0.3,0.1

Type RM Length L Ch R = 1 ,4038    ,226.1,225.8,225.5
XS GIS Cut Line= 4
      1609483.47      247557.982     1609140.635       247341.81
     1608760.406      247462.408     1608529.965      247451.782
#Sta/Elev= 30
    10.1  835.87    30.4  829.75    60.8  823.29    81.1  820.19    91.2  817.88
   101.3  814.31   162.1  784.47   172.3   778.9   182.4  771.36   202.6  758.54
   212.8  755.33   344.5  748.81   415.3  747.43   455.2   741.5   475.1  735.79
   534.9  731.01   674.6  733.22   684.5  732.69   704.4  726.42   714.4     726
  721.34  727.02   774.3  740.19   804.2  744.48   834.3  755.05   854.3  766.97
   904.5  787.46   924.6  799.22   984.7  822.63  1004.8  834.24  1034.9  845.74
#Mann= 3 , 0 , 0
    10.1     .08       0   704.4    .045       0  721.34     .08       0
#XS Ineff= 2 , 0
       0     672                       0
Permanent Ineff=
       F       F
Bank Sta=704.4,721.34
XS Rating Curve= 0 ,0
Exp/Cntr=0.3,0.1

Type RM Length L Ch R = 1 ,3812.2  ,259.3,255.8,252.3
XS GIS Cut Line= 4
     1609202.043      247009.393     1609038.367      247135.097
     1608687.445      247250.325     1608517.222      247268.656
#Sta/Elev= 30
       0  873.55     9.8  873.55    19.7  865.19    39.3  852.32   167.1  782.82
   176.9  775.58   186.7  766.45   206.4  754.32   216.4  750.13   236.3  746.62
   266.3  744.06   276.3  741.07   296.2  732.29   306.2  729.94   356.1   726.4
   386.1  727.25     446   731.6   455.9  731.27  472.35  726.31   485.9  724.95
  488.78  726.35   555.8  758.95   565.7  767.73   636.2  802.21   646.2  810.64
   656.3  816.41   706.7   839.8   716.7  847.76   726.8  854.13   746.9  863.73
#Mann= 3 , 0 , 0
       0      .1       0  472.35    .045       0  488.78      .1       0
#XS Ineff= 2 , 0
       0     446                       0
Permanent Ineff=
       F       F
Bank Sta=472.35,488.78
XS Rating Curve= 0 ,0
Exp/Cntr=0.3,0.1

Type RM Length L Ch R = 1 ,3556.4  ,182,181.6,181.2
XS GIS Cut Line= 4
     1609042.389      246852.888     1608833.455      246903.415
     1608636.812      247008.564     1608497.523      247154.681
#Sta/Elev= 30
     9.8  830.74    19.5  825.05    87.9  794.27    97.7  787.07   117.2  777.38
   156.3  754.64   166.1  745.92   175.9  742.33     215  740.24   224.7  736.66
   234.3  730.38     244  725.93   263.4  726.14   292.5  720.95   302.2  720.37
   360.4   722.3  374.48  721.42   389.5  719.19  394.09  721.01   399.2  722.93
   418.6  738.81   428.3  744.37   478.3  765.99   498.5  779.06   508.6  783.75
     549  802.26   569.2  808.91   579.3  813.85   599.4  828.59   639.8  848.94
#Mann= 3 , 0 , 0
     9.8     .06       0  374.48    .045       0  394.09     .06       0
Bank Sta=374.48,394.09
XS Rating Curve= 0 ,0
Exp/Cntr=0.3,0.1

Type RM Length L Ch R = 1 ,3374.8  ,264.1,256.8,249.5
XS GIS Cut Line= 4
     1608925.041      246611.677     1608764.813      246730.027
     1608548.141      246852.019     1608424.329      246939.416
#Sta/Elev= 30
      10  835.15    29.9  830.63    79.7  809.63   149.4  762.85   159.4  755.52
   169.3  746.39   179.3  743.03   189.2  741.23     229  739.21     239  735.86
   248.9  728.92   258.9  723.82   278.8  721.81   288.7   719.2   308.6  717.89
   368.3  719.23   378.2  718.59   388.1  716.23   398.1     714   408.1  715.29
     418  723.48     428  729.24   447.9  739.79   488.3  758.43   498.4  765.26
   518.6  772.79   569.1  796.04   579.2  801.24   589.3  808.17   599.4  811.72
#Mann= 3 , 0 , 0
       0     .06       0   388.1    .045       0   408.1     .06       0
Bank Sta=388.1,408.1
XS Rating Curve= 0 ,0
Exp/Cntr=0.3,0.1

Type RM Length L Ch R = 1 ,3118.1  ,185.4,201.7,218
XS GIS Cut Line= 4
     1608718.747      246374.936     1608493.426       246549.73
     1608389.642      246673.998     1608292.686      246858.351
#Sta/Elev= 30
     9.8  827.37    39.3  820.14    78.7  805.65    88.5  800.99    98.3     795
   127.8   770.8   147.5  749.07   157.3   740.1   167.2  733.72   186.8  730.37
   206.5  730.04   216.3  728.29     236  717.97   265.5  718.15   305.4  715.15
   366.1  714.82   386.5  711.86   396.5  709.35   406.5  710.21   416.7  715.92
   426.8  724.46     437  726.77     457  737.13   496.7  755.45   526.4   770.9
   546.3  782.86   556.2  785.46   585.9  801.08   645.5  830.31   655.4  832.07
#Mann= 3 , 0 , 0
       0     .06       0   386.5    .045       0   406.5     .06       0
Bank Sta=386.5,406.5
XS Rating Curve= 0 ,0
Exp/Cntr=0.3,0.1

Type RM Length L Ch R = 1 ,2916.4  ,275.3,270,264.6
XS GIS Cut Line= 4
     1608606.086      246278.321       1608379.4      246480.427
     1608276.982      246491.352     1608076.242      246634.737
#Sta/Elev= 30
    10.1  836.43    30.4  822.22    70.9   800.8    91.1  788.34   111.4  774.43
   121.5  764.15   131.6  757.51   141.7   754.5   151.8  748.42     162  739.93
   172.1  728.88   182.2  724.04   202.5  721.39   232.8  711.99   322.4   713.9
   341.2  712.27   359.2  708.37   369.2  707.14   379.2  708.64   397.3  712.38
   426.4  713.39   436.3  716.14   475.8  734.86   485.6  738.52   505.4  742.96
   525.1  750.25   623.8  801.85   633.7  805.11   643.5  806.43   653.4  810.25
#Mann= 3 , 0 , 0
       0     .06       0   359.2    .045       0   379.2     .06       0
Bank Sta=359.2,379.2
XS Rating Curve= 0 ,0
Exp/Cntr=0.3,0.1

Type RM Length L Ch R = 1 ,2646.5  ,330.8,324.7,317.3
XS GIS Cut Line= 4
     1608588.334      246242.816     1608327.508      246227.795
     1608130.865      246306.998     1608021.619      246611.522
#Sta/Elev= 30
      10  833.56    70.3  810.72    90.4  798.66   130.6  781.11   160.8  763.11
   190.9   750.7   221.1  740.66   231.1   734.4   241.2  725.42   251.2  719.55
   261.3  715.92   271.4  713.98   301.6  712.99   311.7  709.44   331.9  706.47
   372.4  704.21   382.4  703.47   392.4  703.68   463.2   710.5   513.7  711.61
     544  715.68   564.2  716.71   584.5  721.71   594.6  722.75   655.2  741.56
   675.5  750.04   695.7  760.36   705.8  760.23   756.3  788.65   796.8  807.18
#Mann= 3 , 0 , 0
       0     .06       0   372.4    .045       0   392.4     .06       0
Bank Sta=372.4,392.4
XS Rating Curve= 0 ,0
Exp/Cntr=0.3,0.1

Type RM Length L Ch R = 1 ,2321.7  ,385.6,383.8,382
XS GIS Cut Line= 4
      1608320.68      245850.895     1608156.811       245957.41
     1608042.102      246043.442     1607829.072      246233.257
#Sta/Elev= 30
     9.8  838.82    48.9  829.98    58.6  826.17    78.2  815.74      88   809.1
    97.7  800.99   117.3  790.06   146.6  777.56   166.1  766.43   185.7  750.09
   233.7  717.57   252.8  702.63   261.9  697.56   271.9   696.9   281.9  697.78
     291  701.35   300.6   703.9   329.3  703.89   437.2  701.59   506.1  705.33
   515.9  707.82   525.8   714.7   535.6  724.95   545.4  731.73   565.1   740.4
     575  746.91   584.8  752.38   604.5  761.39   614.3  766.73   624.2  774.67
#Mann= 3 , 0 , 0
       0     .08       0   261.9    .045       0   281.9     .08       0
Bank Sta=261.9,281.9
XS Rating Curve= 0 ,0
Exp/Cntr=0.3,0.1

Type RM Length L Ch R = 1 ,1937.9  ,369.1,364.3,359.6
XS GIS Cut Line= 4
     1608125.403       245543.64     1607911.007      245656.983
     1607762.159       245790.81     1607591.461      245990.184
#Sta/Elev= 30
    10.1  851.65    60.6  836.54    70.7  832.32    80.8  825.94   121.3  811.07
   151.6  797.04   161.7  789.45   171.8  783.36   232.4  754.56   252.5  740.87
   262.5  735.08   272.5   732.4   282.5  727.62   312.6  708.94   332.6     691
   342.6   690.3   352.6  690.88   422.7  695.38   483.1  696.41   503.2  699.23
   523.4  703.77   533.5  707.58   543.6  709.86     584  727.69   604.2  737.61
   614.3  743.33   624.4  750.75   644.6  761.57   664.8  768.16   705.1  787.93
#Mann= 3 , 0 , 0
       0     .08       0   332.6    .045       0   352.6     .08       0
Bank Sta=332.6,352.6
XS Rating Curve= 0 ,0
Exp/Cntr=0.3,0.1

Type RM Length L Ch R = 1 ,1573.6  ,379.3,381.4,383.5
XS GIS Cut Line= 4
     1607678.858      245224.095     1607613.311      245424.835
     1607494.985       245596.58     1607407.108      245824.949
#Sta/Elev= 30
    10.1  834.83    20.1  831.54    60.3  803.38    90.5  784.63   110.6  770.44
   120.7  769.19   130.7  763.37   211.2  710.26   221.1   704.7     231  702.93
     241   696.3   250.9  687.56   260.8  683.09   270.8  682.81   280.8  683.03
   320.4  684.46   350.2  684.85   419.7  691.09   429.5  691.66   458.9  691.81
   468.7  692.57   488.2  696.63     498   699.9   507.8  705.01     547   729.9
   556.8   730.8   595.9  756.29   605.7  761.58   654.6  785.67   664.4  787.08
#Mann= 3 , 0 , 0
       0      .1       0   260.8    .045       0   280.8     .06       0
Bank Sta=260.8,280.8
XS Rating Curve= 0 ,0
Exp/Cntr=0.3,0.1

Type RM Length L Ch R = 1 ,1192.2  ,259.9,267.7,275.6
XS GIS Cut Line= 4
     1607463.097      244989.215     1607285.572      245241.847
     1607176.326      245370.212     1607105.795      245402.668
#Sta/Elev= 30
      10  881.76    19.9  880.36    29.9  876.44    49.8  868.21    59.8  863.72
    79.7  853.63    89.6  848.29    99.6  842.64   109.6  836.68   119.5   829.2
   129.5  825.59   139.4  820.01   149.4  813.22   189.2  787.92   209.2  775.02
   219.1  768.47   229.1  759.98     239   752.2     249  748.54     259  745.36
   288.8   725.6   318.7   705.1   328.6  696.48   338.5   686.8   348.3  682.87
   358.3  682.43   368.3   682.5   516.1   687.2   535.6  687.54     555  687.56
#Mann= 3 , 0 , 0
       0      .1       0   348.3    .045       0   368.3     .06       0
Bank Sta=348.3,368.3
XS Rating Curve= 0 ,0
Exp/Cntr=0.3,0.1

Type RM Length L Ch R = 1 ,924.5   ,214,217.1,220.2
XS GIS Cut Line= 4
     1607357.948      244878.603     1607165.401      245047.935
     1606981.527      245141.842     1606944.657      245163.691
#Sta/Elev= 30
     9.9  879.74    19.7  878.09    39.4   873.6    59.2  870.38      69  866.75
    78.9  858.72    88.8   853.4   118.3  839.07   147.9  823.21   157.8  819.49
   167.7  810.37   177.5   802.9   197.2  791.67   226.8  775.38   236.7  769.25
   246.6  759.55   256.4  746.58   266.2  739.87   276.1  733.64   295.7  719.49
   325.2  704.01   335.1  694.73   354.7  683.46   364.4   679.4   374.4  677.96
   384.4  678.14   462.9  682.46   471.4  682.81   497.2  682.81   505.7  683.17
#Mann= 3 , 0 , 0
       0      .1       0   364.4    .045       0   384.4     .06       0
Bank Sta=364.4,384.4
XS Rating Curve= 0 ,0
Exp/Cntr=0.3,0.1

Type RM Length L Ch R = 1 ,707.4   ,270.7,270.3,269.9
XS GIS Cut Line= 4
     1607338.829      244841.733     1607064.348      244874.507
     1606815.813      244956.441     1606541.332      245015.161
#Sta/Elev= 30
     9.9  880.27    39.5  870.75    59.2  857.94   108.6  830.98   128.3  814.95
   148.1  804.32   177.7  790.38   187.6  783.88   197.5  774.89   266.6   738.8
   276.4  729.85   336.8  700.73     357  683.93     367  678.12   377.1  675.36
   387.1  675.28   397.1  675.89   447.5  678.15   487.8  678.51   598.3  689.37
   618.3  693.59   638.4  702.28   648.4   708.6   658.4  719.08   718.6  749.73
   728.6  757.11   788.7  781.23   798.8  787.92   808.8  792.97   818.8  796.16
#Mann= 3 , 0 , 0
       0      .1       0   377.1    .045       0   397.1     .06       0
Bank Sta=377.1,397.1
XS Rating Curve= 0 ,0
Exp/Cntr=0.3,0.1

Type RM Length L Ch R = 1 ,437.1   ,344.2,352.5,360.7
XS GIS Cut Line= 4
     1607340.863      244663.949     1607033.588      244596.442
     1606591.298      244752.407      1606363.17      244796.636
#Sta/Elev= 30
       0  890.06     9.8  890.06    78.7  855.68   137.6  835.09   147.5  827.16
   216.3  796.59     236  783.74   304.8  754.98   314.6  748.31   374.5  719.86
   394.4  706.62   444.3  684.51   454.3  679.07   464.3  668.87  470.13  667.72
   474.3  666.93  489.26  667.86   544.1  673.86   663.8  679.61   683.8  682.94
   713.7  693.84   753.7  713.06   763.6  719.23   783.6   738.4   834.1  764.81
   854.3  779.98   904.8  806.29     925  821.34   985.7  850.58    1016  867.46
#Mann= 3 , 0 , 0
       0      .1       0  470.13    .045       0  489.26     .06       0
Bank Sta=470.13,489.26
XS Rating Curve= 0 ,0
Exp/Cntr=0.3,0.1

Type RM Length L Ch R = 1 ,84.6    ,86.9,84.6,82.3
XS GIS Cut Line= 4
     1607294.306      244338.051      1606912.54      244319.429
     1606486.545      244289.167     1606188.582      244233.298
#Sta/Elev= 30
       0  951.31    10.1  951.31    40.2  934.32    60.4  918.63   120.7  892.36
   140.8  875.59   160.9  863.87   191.1  852.98   201.2  847.04   211.2  835.71
   291.7  788.83     352   758.1   362.1  747.12   431.9  707.95   451.7  691.31
   491.5  669.55  509.98  665.39   521.3  665.06  529.69  665.37     700  675.57
   729.8  682.94   809.3  726.98   819.4  738.51   890.1  776.05   910.3  791.58
   960.9   817.4   991.2  838.96  1041.7  864.86  1061.9   881.1  1112.4  907.38
#Mann= 3 , 0 , 0
       0      .1       0  509.98    .045       0  529.69     .06       0
Bank Sta=509.98,529.69
XS Rating Curve= 0 ,0
Exp/Cntr=0.3,0.1
Stream Node=sycmrcrk        ,Main            , 0 , 0 ,Upstream end
Stream Node=sycmrcrk        ,Main            , 0 , 1 ,Downstream end

Chan Stop Cuts=-1
Use User Specified Reach Order=0
